HEC-RAS study ras_bridge.prj: ras_bridge

--- ras_bridge.g01 (geometry) --- (continued)

Type RM Length L Ch R = 3 ,500     ,,,
Bridge Culvert--1,0,-1,-1, 0
Deck Dist Width WeirC Skew NumUp NumDn MinLoCord MaxHiCord MaxSubmerge Is_Ogee
15,20,1.4,0, 6, 6, , , 0.98, 0, 0,0,,
       0      10   10.01   19.99      20      30
      -1      -1      -1      -1      -1      -1
    -2.5    -2.5    -2.2    -2.2    -2.5    -2.5
       0      10   10.01   19.99      20      30
      -1      -1      -1      -1      -1      -1
    -2.7    -2.7    -2.2    -2.2    -2.7    -2.7
BR Coef=-1 , 0 , 0 ,, 0 ,,,0.8,-1,,0,
WSPro=,,,, 1 ,,,, 0 ,,,, 0 ,,,,-1 ,-1 ,-1 , 0 , 0 , 0 , 0 , 0
BC Design=,, 0 ,, 0 ,,,,,,
BC HTab HWMax=3
BC HTab TWMax=3
BC Use User HTab Curves=0
BC User HTab FreeFlow(D)= 100
              0.          -3.372            0.05          -3.316
           0.125          -3.278             0.3          -3.227
           0.499          -3.181           0.749          -3.139
           0.998          -3.102           1.248           -3.07
           1.498           -3.04           1.747          -3.012
           1.997          -2.987           2.247          -2.962
           2.496           -2.94           2.746          -2.918
           2.995          -2.897           3.245          -2.878
           3.495          -2.859           3.744          -2.841
           3.994          -2.823           4.243          -2.806
           4.493          -2.789           4.743          -2.773
           4.992          -2.757           5.242          -2.741
           5.492          -2.725           5.741           -2.71
           5.991          -2.696            6.24          -2.682
            6.49          -2.668            6.74          -2.654
           6.989          -2.639           7.239          -2.626
           7.489          -2.613           7.738          -2.599
           7.988          -2.586           8.237          -2.572
           8.487          -2.559           8.737          -2.548
           8.986          -2.537           9.236          -2.525
           9.485          -2.515           9.735          -2.504
           9.985          -2.493          10.234          -2.483
          10.484          -2.472          10.734          -2.461
          10.983          -2.451          11.233           -2.44
          11.482           -2.43          11.732          -2.419
          13.514          -2.337          15.295          -2.259
          17.077          -2.053          18.858          -1.935
           20.64          -1.818          22.421          -1.697
          24.203          -1.562          25.984          -1.424
          27.766          -1.282          29.547          -1.138
          32.896          -0.853          36.624          -0.504
          40.774          -0.104          45.395          -0.104
          50.539          -0.104          56.266          -0.063
          62.642           0.011          69.741            0.09
          77.645           0.174          86.444           0.265
           96.24           0.363         107.146           0.467
         119.288           0.578         132.806           0.697
         147.856           0.824         164.612           0.959
         183.266           1.104         204.035           1.258
         227.157           1.422         252.899           1.596
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BC User HTab Sub Curve(D)= 47
              0.          -3.168           0.016          -3.168
           0.032          -3.168           0.048          -3.168
           0.064          -3.167            0.08          -3.167
           0.096          -3.167           0.112          -3.167
           0.128          -3.166           0.144          -3.166
            0.16          -3.166           0.176          -3.165
           0.192          -3.165           0.208          -3.164
           0.224          -3.163            0.24          -3.163
           0.256          -3.162           0.272          -3.162
           0.288          -3.161           0.304           -3.16
            0.32          -3.159           0.336          -3.158
           0.352          -3.158           0.368          -3.157
           0.384          -3.156             0.4          -3.155
           0.416          -3.154           0.432          -3.153
           0.448          -3.152           0.464          -3.151
            0.48          -3.149           0.496          -3.148
           0.512          -3.147           0.528          -3.146
           0.544          -3.145            0.56          -3.143
           0.576          -3.142           0.592          -3.141
           0.608           -3.14           0.624          -3.138
            0.64          -3.137           0.656          -3.135
           0.672          -3.134           0.688          -3.133
           0.704          -3.131            0.72           -3.13
           0.811           -3.13
BC User HTab Sub Curve(D)= 45
              0.          -2.963            0.07          -2.963
           0.139          -2.963           0.209          -2.963
           0.278          -2.963           0.348          -2.962
           0.417          -2.962           0.487          -2.961
           0.556          -2.961           0.626           -2.96
           0.695          -2.959           0.765          -2.958
           0.835          -2.957           0.904          -2.956
           0.974          -2.955           1.043          -2.953
           1.113          -2.952           1.182          -2.951
           1.252          -2.949           1.321          -2.947
           1.391          -2.946           1.461          -2.944
            1.53          -2.942             1.6           -2.94
           1.669          -2.938           1.739          -2.936
           1.808          -2.934           1.878          -2.932
           1.947          -2.929           2.017          -2.927
           2.086          -2.924           2.156          -2.922
           2.226          -2.919           2.295          -2.916
           2.365          -2.913           2.434           -2.91
           2.504          -2.907           2.573          -2.904
           2.643          -2.901           2.712          -2.898
           2.782          -2.895           2.851          -2.891
           2.921          -2.888           2.991          -2.885
           3.162          -2.885
BC User HTab Sub Curve(D)= 39
              0.          -2.759            0.18          -2.759
           0.361          -2.759           0.541          -2.758
           0.722          -2.758           0.902          -2.757
           1.083          -2.756           1.263          -2.755
           1.444          -2.754           1.624          -2.753
           1.805          -2.751           1.985           -2.75
           2.166          -2.748           2.346          -2.746
           2.527          -2.744           2.707          -2.741
           2.888          -2.739           3.068          -2.736
           3.249          -2.734           3.429          -2.731
            3.61          -2.727            3.79          -2.724
           3.971           -2.72           4.151          -2.717
           4.332          -2.713           4.512          -2.709
           4.692          -2.704           4.873            -2.7
           5.053          -2.695           5.234           -2.69
           5.414          -2.685           5.595           -2.68
           5.775          -2.675           5.956          -2.669
           6.136          -2.663           6.317          -2.657
           6.497          -2.651           6.678          -2.645
           6.897          -2.645
BC User HTab Sub Curve(D)= 38
              0.          -2.555           0.389          -2.555
           0.778          -2.554           1.166          -2.553
           1.555          -2.552           1.944           -2.55
           2.333          -2.548           2.721          -2.545
            3.11          -2.542           3.499          -2.539
           3.888          -2.535           4.276           -2.53
           4.665          -2.526           5.054          -2.521
           5.443          -2.515           5.831          -2.509
            6.22          -2.503           6.609          -2.496
           6.998          -2.489           7.386          -2.481
           7.775          -2.473           8.164          -2.464
           8.553          -2.455           8.942          -2.446
            9.33          -2.436           9.719          -2.426
          10.108          -2.416          10.497          -2.406
          10.885          -2.395          11.274          -2.383
          11.663          -2.372          12.052          -2.361
           12.44          -2.349          12.829          -2.337
          13.218          -2.326          13.607          -2.313
          13.995          -2.301          14.331          -2.301
BC User HTab Sub Curve(D)= 42
              0.          -2.351           0.534           -2.35
           1.068          -2.349           1.602          -2.348
           2.136          -2.345            2.67          -2.342
           3.204          -2.339           3.738          -2.334
           4.272          -2.329           4.806          -2.323
            5.34          -2.317           5.874           -2.31
           6.408          -2.302           6.942          -2.293
           7.476          -2.283            8.01          -2.273
           8.544          -2.262           9.078          -2.251
           9.612          -2.238          10.146          -2.225
           10.68          -2.211          11.214          -2.196
          11.748           -2.18          12.282          -2.164
          12.816          -2.146           13.35          -2.128
          13.884          -2.109          14.418          -2.089
          14.952          -2.068          15.486          -2.047
           16.02          -2.025          16.554          -2.001
          17.088          -1.978          17.622          -1.953
          18.156          -1.928           18.69          -1.901
          19.224          -1.874          19.758          -1.846
          20.292          -1.816          20.826          -1.786
           21.36          -1.755          21.558          -1.755
BC User HTab Sub Curve(D)= 43
              0.          -2.146           0.694          -2.146
           1.388          -2.144           2.081          -2.142
           2.775          -2.138           3.469          -2.134
           4.163          -2.128           4.856          -2.122
            5.55          -2.114           6.244          -2.105
           6.938          -2.096           7.632          -2.085
           8.325          -2.073           9.019           -2.06
           9.713          -2.046          10.407          -2.031
          11.101          -2.014          11.794          -1.997
          12.488          -1.979          13.182          -1.959
          13.876          -1.938          14.569          -1.916
          15.263          -1.893          15.957          -1.869
          16.651          -1.843          17.345          -1.816
          18.038          -1.788          18.732          -1.759
          19.426          -1.729           20.12          -1.697
          20.814          -1.664          21.507           -1.63
          22.201          -1.595          22.895          -1.558
          23.589          -1.521          24.282          -1.481
          24.976          -1.441           25.67          -1.399
          26.364          -1.357          27.058          -1.312
          27.751          -1.267          28.445           -1.22
          28.532           -1.22
BC User HTab Sub Curve(D)= 43
              0.          -1.942           0.867          -1.941
           1.734          -1.939           2.601          -1.936
           3.468           -1.93           4.334          -1.924
           5.201          -1.916           6.068          -1.906
           6.935          -1.896           7.802          -1.883
           8.669          -1.869           9.536          -1.854
          10.403          -1.837           11.27          -1.818
          12.137          -1.798          13.003          -1.776
           13.87          -1.753          14.737          -1.728
          15.604          -1.701          16.471          -1.673
          17.338          -1.643          18.205          -1.612
          19.072          -1.578          19.939          -1.543
          20.806          -1.507          21.672          -1.468
          22.539          -1.428          23.406          -1.386
          24.273          -1.343           25.14          -1.297
          26.007           -1.25          26.874          -1.201
          27.741           -1.15          28.608          -1.097
          29.475          -1.042          30.341          -0.986
          31.208          -0.927          32.075          -0.866
          32.942          -0.801          33.809          -0.734
          34.676          -0.665          35.543          -0.595
          35.648          -0.595
BC User HTab Sub Curve(D)= 42
              0.          -1.738           1.052          -1.737
           2.104          -1.734           3.157          -1.729
           4.209          -1.722           5.261          -1.713
           6.313          -1.701           7.365          -1.688
           8.417          -1.673            9.47          -1.656
          10.522          -1.636          11.574          -1.615
          12.626          -1.591          13.678          -1.565
          14.731          -1.537          15.783          -1.507
          16.835          -1.474          17.887          -1.439
          18.939          -1.402          19.992          -1.363
          21.044          -1.321          22.096          -1.277
          23.148          -1.231            24.2          -1.182
          25.252          -1.131          26.305          -1.077
          27.357           -1.02          28.409          -0.961
          29.461            -0.9          30.513          -0.834
          31.566          -0.765          32.618          -0.693
           33.67           -0.62          34.722          -0.543
          35.774          -0.464          36.827          -0.383
          37.879          -0.299          38.931          -0.214
          39.983          -0.126          41.035          -0.037
          42.087          -0.037          58.508          -0.037
BC User HTab Sub Curve(D)= 38
              0.          -1.533           1.248          -1.532
           2.496          -1.528           3.743          -1.521
           4.991          -1.512           6.239          -1.499
           7.487          -1.484           8.734          -1.466
           9.982          -1.446           11.23          -1.422
          12.478          -1.396          13.725          -1.367
          14.973          -1.334          16.221          -1.299
          17.469          -1.261          18.716           -1.22
          19.964          -1.176          21.212          -1.128
           22.46          -1.078          23.707          -1.024
          24.955          -0.967          26.203          -0.907
          27.451          -0.842          28.698          -0.772
          29.946            -0.7          31.194          -0.625
          32.442          -0.545          33.689          -0.463
          34.937          -0.377          36.185          -0.289
          37.433          -0.197           38.68          -0.102
          39.928          -0.005          41.176           0.096
          42.424           0.096          58.508           0.096
          69.741           0.096           70.28           0.096
BC User HTab Sub Curve(D)= 46
              0.          -1.329            0.97          -1.328
            1.94          -1.326            2.91          -1.322
            3.88          -1.316           4.851          -1.309
           5.821            -1.3           6.791           -1.29
           7.761          -1.278           8.731          -1.264
           9.701          -1.249          10.671          -1.231
          11.641          -1.213          12.611          -1.192
          13.582           -1.17          14.552          -1.146
          15.522          -1.121          16.492          -1.094
          17.462          -1.065          18.432          -1.034
          19.402          -1.001          20.372          -0.967
          21.342           -0.93          22.312          -0.892
          23.283          -0.852          24.253          -0.809
          25.223          -0.764          26.193          -0.717
          27.163          -0.669          28.133          -0.618
          29.103          -0.565          30.073          -0.511
          31.043          -0.454          32.014          -0.396
          32.984          -0.336          33.954          -0.274
          34.924           -0.21          35.894          -0.145
          36.864          -0.077          37.834          -0.008
          38.804           0.063          39.774           0.135
          40.745            0.21          41.715            0.21
           70.28            0.21          81.079            0.21
BC User HTab Sub Curve(D)= 42
              0.          -1.125             1.1          -1.124
             2.2          -1.121             3.3          -1.116
             4.4          -1.109             5.5          -1.099
             6.6          -1.088             7.7          -1.075
             8.8           -1.06             9.9          -1.042
             11.          -1.023            12.1          -1.001
            13.2          -0.977            14.3          -0.951
            15.4          -0.923            16.5          -0.893
            17.6           -0.86            18.7          -0.825
            19.8          -0.788            20.9          -0.748
             22.          -0.705            23.1          -0.661
            24.2          -0.614            25.3          -0.564
            26.4          -0.512            27.5          -0.458
            28.6          -0.402            29.7          -0.343
            30.8          -0.282            31.9          -0.218
             33.          -0.152            34.1          -0.084
            35.2          -0.014            36.3           0.059
            37.4           0.133            38.5            0.21
            39.6            0.29            40.7           0.371
            41.8           0.371          81.079           0.371
           96.24           0.371          97.076           0.371
BC User HTab Sub Curve(D)= 69
              0.          -0.921           0.858           -0.92
           1.716          -0.918           2.575          -0.915
           3.433          -0.911           4.291          -0.905
           5.149          -0.899           6.008          -0.891
           6.866          -0.882           7.724          -0.872
           8.582          -0.861            9.44           -0.85
          10.299          -0.838          11.157          -0.826
          12.015          -0.812          12.873          -0.799
          13.731          -0.785           14.59           -0.77
          15.448          -0.756          16.306          -0.741
          17.164          -0.726          18.023           -0.71
          18.881          -0.694          19.739          -0.678
          20.597          -0.662          21.455          -0.646
          22.314          -0.629          23.172          -0.612
           24.03          -0.596          24.888          -0.579
          25.033          -0.573          25.746           -0.54
          25.811          -0.537          26.605          -0.499
          26.666          -0.496          27.463          -0.457
          27.525          -0.454          28.321          -0.413
           28.38           -0.41          29.179          -0.368
          29.236          -0.365          30.038          -0.321
          30.092          -0.318          30.896          -0.273
          30.948           -0.27          31.754          -0.223
          31.806           -0.22          32.612          -0.172
          32.663          -0.169           33.47           -0.12
          33.519          -0.117          34.329          -0.067
          34.376          -0.064          35.187          -0.012
          35.234          -0.009          36.045           0.045
          36.091           0.048          36.903           0.103
          36.948           0.106          37.762           0.162
          37.805           0.165           38.62           0.222
          38.662           0.225          39.478           0.284
          39.521           0.287            39.6           0.291
            40.7           0.373          97.076           0.374
          97.396           0.374
BC User HTab Sub Curve(D)= 55
              0.          -0.716           1.189          -0.716
           2.377          -0.715           3.566          -0.712
           4.754          -0.709           5.943          -0.705
           7.132            -0.7            8.32          -0.695
           9.509          -0.688          10.697           -0.68
          11.886          -0.671          13.074          -0.661
          14.263          -0.649          15.452          -0.636
           16.64          -0.621          17.829          -0.601
          19.017          -0.562          20.206          -0.523
          21.395          -0.503          22.583          -0.482
          23.772           -0.46           24.96          -0.438
          26.149          -0.415          27.338          -0.391
          28.526          -0.366          29.672          -0.338
          29.715          -0.336          29.798          -0.331
          30.903           -0.27          30.956          -0.266
          32.092            -0.2          32.143          -0.197
          33.281          -0.129           33.33          -0.126
          34.469          -0.055          34.516          -0.052
          35.658           0.022          35.704           0.025
          36.846           0.102          36.891           0.105
          38.035           0.184          38.078           0.187
          39.223           0.269          39.265           0.272
          40.412           0.354          40.453           0.357
            40.7           0.374          41.601           0.376
          42.789           0.376          43.978           0.376
          45.166           0.376          46.355           0.376
          47.544           0.376          97.396           0.377
          97.716           0.377
BC User HTab Sub Curve(D)= 56
              0.          -0.512           1.288          -0.512
           2.577          -0.511           3.865           -0.51
           5.154          -0.509           6.442          -0.507
           7.731          -0.505           9.019          -0.502
          10.308          -0.499          11.596          -0.496
          12.885          -0.492          14.173          -0.487
          15.462          -0.483           16.75          -0.477
          18.038          -0.472          19.327          -0.465
          20.615          -0.458          21.904          -0.451
          23.192          -0.444          24.481          -0.435
          25.534          -0.424          25.769          -0.419
           25.95          -0.416          27.058          -0.394
          27.209          -0.391          28.346          -0.367
          28.492          -0.364          29.635          -0.336
          29.757           -0.33          30.923          -0.265
          30.975          -0.262          32.212           -0.19
          32.262          -0.187            33.5          -0.112
          33.549          -0.109          34.788          -0.031
          34.835          -0.028          36.077           0.053
          36.122           0.056          37.365           0.141
          37.409           0.144          38.654           0.231
          38.696           0.234          39.942           0.324
          39.984           0.327          40.412           0.356
          40.453           0.359            40.7           0.376
          41.231           0.378          42.519           0.379
          43.808           0.379          45.096           0.379
          46.385           0.379          47.673           0.379
          97.716            0.38          98.036            0.38
BC User HTab Sub Curve(D)= 63
              0.          -0.308           0.908          -0.308
           1.817          -0.308           2.725          -0.307
           3.634          -0.307           4.542          -0.307
            5.45          -0.306           6.359          -0.305
           7.267          -0.305           8.176          -0.304
           9.084          -0.303           9.992          -0.302
          10.901          -0.301          11.809          -0.299
          12.718          -0.298          13.626          -0.297
          14.534          -0.295          15.443          -0.294
          16.351          -0.292           17.26           -0.29
          18.168          -0.288          19.077          -0.286
          19.985          -0.284          20.893          -0.281
          21.802          -0.279           22.71          -0.276
          23.619          -0.274          24.527          -0.271
          25.435          -0.268          26.344          -0.265
          27.252          -0.262          28.161          -0.259
          29.069          -0.255          29.977          -0.252
          30.886          -0.248          31.263          -0.242
          31.794          -0.211          31.846          -0.208
          32.703          -0.157          32.753          -0.154
          33.611          -0.102          33.659          -0.099
          34.519          -0.045          34.568          -0.042
          35.428           0.014          35.474           0.017
          36.336           0.074          36.381           0.077
          37.245           0.136          37.289           0.139
          38.153           0.199          38.196           0.202
          39.061           0.263          39.104           0.266
           39.97           0.329          40.012           0.332
          40.412           0.357          40.453            0.36
            40.7           0.377          41.231            0.38
          42.519            0.38          98.036           0.383
          98.355           0.383
BC User HTab Sub Curve(D)= 52
              0.          -0.103           1.785          -0.103
            3.57          -0.103           5.355          -0.102
            7.14          -0.102           8.926          -0.101
          10.711            -0.1          12.496          -0.098
          14.281          -0.097          16.066          -0.095
          17.851          -0.093          19.636           -0.09
          21.421          -0.088          23.206          -0.085
          24.991          -0.082          26.777          -0.079
          28.562          -0.075          30.347          -0.071
          32.132          -0.067          33.917          -0.063
          34.246          -0.059          35.702           0.035
          35.748           0.038          37.487           0.156
          37.531           0.159          39.272           0.282
          39.314           0.285           39.97            0.33
          40.012           0.333          40.412           0.359
          40.453           0.362            40.7           0.379
          41.057           0.382          41.722           0.385
          42.842           0.385          44.628           0.385
          46.413           0.385          48.198           0.385
          49.983           0.385          51.768           0.385
          53.553           0.385          55.338           0.385
          57.123           0.385          58.908           0.385
          60.694           0.385          62.479           0.385
          64.264           0.385          66.049           0.385
          67.834           0.385          69.619           0.385
          98.355           0.386          98.675           0.386
BC User HTab Sub Curve(D)= 57
              0.           0.101            2.09           0.101
           4.181           0.101           6.271           0.102
           8.361           0.102          10.452           0.103
          12.542           0.104          14.632           0.105
          16.723           0.107          18.813           0.108
          20.903            0.11          22.994           0.112
          25.084           0.114          27.174           0.117
          29.265           0.119          31.355           0.122
          33.445           0.125          35.536           0.128
          37.189           0.138          37.626           0.168
          37.669           0.171          39.716           0.316
           39.76           0.319           39.97           0.332
          40.012           0.335          40.412            0.36
          40.453           0.363            40.7            0.38
          41.057           0.383          41.807           0.388
          43.897           0.388          45.987           0.388
          48.078           0.388          50.168           0.388
          52.258           0.388          54.349           0.388
          56.439           0.388          58.529           0.388
           60.62           0.388           62.71           0.388
            64.8           0.388          66.891           0.388
          68.981           0.388          71.071           0.388
          73.162           0.388          75.252           0.388
          77.342           0.388          79.433           0.388
          81.523           0.389          83.613           0.389
          85.704           0.389          87.794           0.389
          89.884           0.389          91.975           0.389
          94.065           0.389          98.675           0.389
          98.995           0.389
BC User HTab Sub Curve(D)= 42
              0.           0.305           3.647           0.305
           7.295           0.306          10.942           0.307
          14.589           0.308          18.237            0.31
          21.884           0.312          25.531           0.314
          29.179           0.317          32.826           0.321
          36.473           0.325          39.968           0.335
           40.12           0.345          40.168           0.348
          40.412           0.362          40.453           0.365
            40.7           0.382          41.057           0.385
          41.807           0.389          43.768           0.391
          47.415           0.391          51.062           0.391
           54.71           0.391          58.357           0.391
          62.004           0.391          65.652           0.391
          69.299           0.391          72.946           0.391
          76.594           0.401          80.241           0.412
          83.888           0.423          87.536           0.436
          91.183           0.448           94.83           0.463
          98.478           0.478         102.125           0.494
         105.772           0.511          109.42            0.53
         113.067            0.55         116.714           0.572
         119.288           0.588         120.473           0.588
BC User HTab Sub Curve(D)= 37
              0.           0.509           4.198            0.51
           8.396            0.51          12.594           0.511
          16.792           0.512           20.99           0.514
          25.188           0.516          29.386           0.518
          33.584           0.521          37.782           0.524
           41.98           0.528          46.178           0.532
          50.376           0.536          54.574           0.541
          58.772           0.546           62.97           0.552
          67.167           0.558          71.365           0.565
          75.563           0.573          79.761           0.581
          83.959            0.59          88.157           0.599
          92.355           0.609          96.553            0.62
         100.751           0.631         104.949           0.644
         109.147           0.656         113.345            0.67
         117.543           0.686         121.741           0.702
         125.939           0.719         130.137           0.737
         134.335           0.757         138.533           0.778
         142.731           0.801         146.929           0.825
         148.024           0.825
BC User HTab Sub Curve(D)= 39
              0.           0.714           4.785           0.714
            9.57           0.714          14.356           0.715
          19.141           0.716          23.926           0.718
          28.711            0.72          33.497           0.722
          38.282           0.725          43.067           0.728
          47.852           0.731          52.638           0.735
          57.423           0.739          62.208           0.744
          66.993           0.749          71.779           0.754
          76.564            0.76          81.349           0.766
          86.134           0.774           90.92           0.782
          95.705            0.79          100.49           0.799
         105.275           0.808         110.061           0.819
         114.846            0.83         119.631           0.841
         124.416           0.854         129.202           0.867
         133.987           0.881         138.772           0.897
         143.557           0.913         148.343            0.93
         153.128           0.949         157.913           0.969
         162.698            0.99         167.484           1.013
         172.269           1.038         177.054           1.064
         178.126           1.064
BC User HTab Sub Curve(D)= 40
              0.           0.918           5.416           0.918
          10.832           0.919          16.248           0.919
          21.664           0.921           27.08           0.922
          32.495           0.924          37.911           0.926
          43.327           0.929          48.743           0.931
          54.159           0.935          59.575           0.938
          64.991           0.942          70.407           0.947
          75.823           0.952          81.239           0.957
          86.655           0.963           92.07           0.969
          97.486           0.976         102.902           0.983
         108.318           0.992         113.734              1.
          119.15           1.009         124.566           1.019
         129.982            1.03         135.398           1.041
         140.814           1.053         146.229           1.066
         151.645            1.08         157.061           1.095
         162.477           1.111         167.893           1.128
         173.309           1.146         178.725           1.165
         184.141           1.186         189.557           1.208
         194.973           1.231         200.389           1.257
         205.804           1.284         207.687           1.284
BC User HTab Sub Curve(D)= 42
              0.           1.122           6.076           1.122
          12.153           1.123          18.229           1.124
          24.305           1.125          30.381           1.126
          36.458           1.128          42.534            1.13
           48.61           1.133          54.686           1.135
          60.763           1.139          66.839           1.142
          72.915           1.146          78.992            1.15
          85.068           1.155          91.144            1.16
           97.22           1.166         103.297           1.172
         109.373           1.179         115.449           1.186
         121.525           1.194         127.602           1.202
         133.678           1.211         139.754           1.221
         145.831           1.231         151.907           1.242
         157.983           1.254         164.059           1.267
         170.136            1.28         176.212           1.295
         182.288            1.31         188.364           1.326
         194.441           1.344         200.517           1.363
         206.593           1.383         212.669           1.404
         218.746           1.427         224.822           1.452
         230.898           1.478         236.975           1.506
         243.051           1.537         244.168           1.537
BC User HTab Sub Curve(D)= 43
              0.           1.327            6.77           1.327
          13.539           1.327          20.309           1.328
          27.079           1.329          33.849            1.33
          40.618           1.332          47.388           1.334
          54.158           1.337          60.928           1.339
          67.697           1.342          74.467           1.346
          81.237            1.35          88.006           1.354
          94.776           1.359         101.546           1.364
         108.316           1.369         115.085           1.375
         121.855           1.382         128.625           1.389
         135.395           1.396         142.164           1.405
         148.934           1.414         155.704           1.423
         162.473           1.433         169.243           1.444
         176.013           1.455         182.783           1.468
         189.552           1.481         196.322           1.495
         203.092            1.51         209.862           1.526
         216.631           1.543         223.401           1.562
         230.171           1.581          236.94           1.602
          243.71           1.625          250.48           1.649
          257.25           1.675         264.019           1.703
         270.789           1.732         277.559           1.764
         278.811           1.764
BC User HTab Sub Curve(D)= 44
              0.           1.531           7.489           1.531
          14.978           1.531          22.467           1.532
          29.956           1.533          37.446           1.535
          44.935           1.536          52.424           1.538
          59.913           1.541          67.402           1.543
          74.891           1.546           82.38            1.55
          89.869           1.554          97.359           1.558
         104.848           1.562         112.337           1.567
         119.826           1.573         127.315           1.579
         134.804           1.585         142.293           1.592
         149.782           1.599         157.272           1.608
         164.761           1.616          172.25           1.625
         179.739           1.635         187.228           1.646
         194.717           1.657         202.206           1.669
         209.695           1.682         217.185           1.696
         224.674           1.711         232.163           1.727
         239.652           1.744         247.141           1.762
          254.63           1.781         262.119           1.802
         269.608           1.824         277.098           1.847
         284.587           1.873         292.076             1.9
         299.565           1.929         307.054            1.96
         313.465           1.989         315.044           1.989
BC User HTab Sub Curve(D)= 45
              0.           1.735           8.234           1.735
          16.469           1.736          24.703           1.736
          32.938           1.738          41.172           1.739
          49.407           1.741          57.641           1.743
          65.875           1.745           74.11           1.747
          82.344            1.75          90.579           1.754
          98.813           1.758         107.048           1.762
         115.282           1.766         123.516           1.771
         131.751           1.776         139.985           1.782
          148.22           1.788         156.454           1.795
         164.689           1.802         172.923            1.81
         181.158           1.819         189.392           1.828
         197.626           1.838         205.861           1.848
         214.095           1.859          222.33           1.871
         230.564           1.884         238.799           1.898
         247.033           1.912         255.267           1.928
         263.502           1.944         271.736           1.962
         279.971           1.981         288.205           2.001
          296.44           2.023         304.674           2.047
         312.908           2.071         321.143           2.098
         329.377           2.127         337.612           2.157
         345.846            2.19         348.988           2.203
         351.541           2.203
BC User HTab Sub Curve(D)= 46
              0.           1.939           9.009            1.94
          18.018            1.94          27.026           1.941
          36.035           1.942          45.044           1.943
          54.053           1.945          63.062           1.947
          72.071           1.949          81.079           1.952
          90.088           1.955          99.097           1.958
         108.106           1.962         117.115           1.966
         126.124            1.97         135.132           1.975
         144.141            1.98          153.15           1.986
         162.159           1.992         171.168           1.999
         180.176           2.006         189.185           2.013
         198.194           2.022         207.203           2.031
         216.212            2.04         225.221           2.051
         234.229           2.062         243.238           2.073
         252.247           2.086         261.256           2.099
         270.265           2.114         279.274           2.129
         288.282           2.146         297.291           2.163
           306.3           2.182         315.309           2.202
         324.318           2.223         333.327           2.246
         342.335           2.271         351.344           2.297
         360.353           2.325         369.362           2.355
         378.371           2.388         387.379           2.422
         396.388            2.46         397.607            2.46
BC User HTab Sub Curve(D)= 47
              0.           2.144           9.805           2.144
           19.61           2.144          29.415           2.145
           39.22           2.146          49.025           2.147
          58.829           2.149          68.634           2.151
          78.439           2.153          88.244           2.156
          98.049           2.159         107.854           2.162
         117.659           2.165         127.464           2.169
         137.269           2.174         147.074           2.178
         156.879           2.184         166.683           2.189
         176.488           2.195         186.293           2.202
         196.098           2.209         205.903           2.216
         215.708           2.224         225.513           2.234
         235.318           2.243         245.123           2.253
         254.928           2.264         264.733           2.276
         274.537           2.288         284.342           2.301
         294.147           2.315         303.952           2.331
         313.757           2.347         323.562           2.364
         333.367           2.382         343.172           2.402
         352.977           2.423         362.782           2.446
         372.587            2.47         382.392           2.496
         392.196           2.524         402.001           2.553
         411.806           2.585         421.611           2.619
         431.416           2.656         432.567           2.661
         435.284           2.661
BC User HTab Sub Curve(D)= 47
              0.           2.348          10.626           2.348
          21.253           2.349          31.879           2.349
          42.505            2.35          53.132           2.352
          63.758           2.353          74.384           2.355
          85.011           2.357          95.637            2.36
         106.263           2.363          116.89           2.366
         127.516           2.369         138.142           2.373
         148.769           2.378         159.395           2.382
         170.021           2.387         180.648           2.393
         191.274           2.399           201.9           2.405
         212.527           2.412         223.153            2.42
         233.779           2.428         244.406           2.437
         255.032           2.446         265.658           2.456
         276.285           2.467         286.911           2.478
         297.537            2.49         308.164           2.503
          318.79           2.517         329.416           2.532
         340.043           2.548         350.669           2.565
         361.295           2.584         371.922           2.602
         382.548           2.623         393.174           2.646
         403.801           2.669         414.427           2.695
         425.054           2.723          435.68           2.752
         446.306           2.783         456.933           2.817
         467.559           2.853         478.185           2.892
         480.611           2.892
BC User HTab Sub Curve(D)= 48
              0.           2.552          11.469           2.552
          22.938           2.553          34.406           2.554
          45.875           2.555          57.344           2.556
          68.813           2.557          80.281           2.559
           91.75           2.561         103.219           2.564
         114.688           2.567         126.157            2.57
         137.625           2.573         149.094           2.577
         160.563           2.582         172.032           2.586
         183.501           2.591         194.969           2.596
         206.438           2.602         217.907           2.609
         229.376           2.616         240.844           2.623
         252.313           2.631         263.782            2.64
         275.251           2.649          286.72           2.659
         298.188           2.669         309.657            2.68
         321.126           2.692         332.595           2.705
         344.063           2.719         355.532           2.734
         367.001           2.749          378.47           2.766
         389.939           2.784         401.407           2.803
         412.876           2.823         424.345           2.845
         435.814           2.869         447.283           2.895
         458.751           2.921          470.22            2.95
         481.689           2.981         493.158           3.014
         504.626           3.049         516.095           3.088
         527.564           3.128          529.65           3.128
BC User HTab Sub Curve(D)= 49
              0.           2.757          12.327           2.757
          24.654           2.757          36.981           2.758
          49.308           2.759          61.635            2.76
          73.962           2.762          86.289           2.763
          98.616           2.766         110.943           2.768
          123.27           2.771         135.597           2.774
         147.924           2.777         160.251           2.781
         172.578           2.785         184.905            2.79
         197.232           2.795         209.559             2.8
         221.886           2.806         234.213           2.812
          246.54           2.819         258.867           2.826
         271.194           2.834         283.521           2.843
         295.848           2.851         308.175           2.861
         320.502           2.871         332.829           2.882
         345.156           2.894         357.483           2.907
         369.811            2.92         382.138           2.935
         394.465            2.95         406.792           2.967
         419.119           2.984         431.446           3.003
         443.773           3.023           456.1           3.045
         468.427           3.068         480.754           3.093
         493.081           3.119         505.408           3.147
         517.735           3.178         530.062           3.211
         542.389           3.246         554.716           3.282
         567.043           3.322          579.37           3.365
         580.732           3.365
BC User HTab Sub Curve(D)= 49
              0.           2.961           13.21           2.961
          26.419           2.961          39.629           2.962
          52.839           2.963          66.049           2.964
          79.258           2.966          92.468           2.968
         105.678            2.97         118.887           2.972
         132.097           2.975         145.307           2.978
         158.517           2.981         171.726           2.985
         184.936           2.989         198.146           2.994
         211.355           2.998         224.565           3.004
         237.775           3.009         250.985           3.015
         264.194           3.022         277.404           3.029
         290.614           3.037         303.824           3.045
         317.033           3.054         330.243           3.064
         343.453           3.074         356.662           3.085
         369.872           3.096         383.082           3.108
         396.292           3.122         409.501           3.136
         422.711           3.151         435.921           3.167
          449.13           3.185          462.34           3.203
          475.55           3.223          488.76           3.244
         501.969           3.267         515.179           3.291
         528.389           3.317         541.598           3.345
         554.808           3.375         568.018           3.407
         581.228           3.442         594.437           3.477
         607.647           3.517         620.857           3.559
         624.205           3.559
BC User HTab Sub Curve(D)= 50
              0.           3.165          14.107           3.165
          28.215           3.166          42.322           3.166
          56.429           3.167          70.536           3.168
          84.644            3.17          98.751           3.172
         112.858           3.174         126.966           3.176
         141.073           3.179          155.18           3.182
         169.287           3.185         183.395           3.189
         197.502           3.193         211.609           3.197
         225.717           3.202         239.824           3.207
         253.931           3.213         268.038           3.219
         282.146           3.225         296.253           3.232
          310.36            3.24         324.467           3.248
         338.575           3.257         352.682           3.266
         366.789           3.276         380.897           3.287
         395.004           3.298         409.111            3.31
         423.218           3.323         437.326           3.337
         451.433           3.352          465.54           3.368
         479.648           3.385         493.755           3.403
         507.862           3.422         521.969           3.443
         536.077           3.465         550.184           3.489
         564.291           3.515         578.399           3.542
         592.506           3.571         606.613           3.603
          620.72           3.636         634.828           3.672
         648.935           3.711         663.042           3.752
          677.15           3.796         679.199           3.796
BC User HTab Sub Curve(D)= 27
              0.           3.369          30.082            3.37
          60.164           3.372          90.245           3.374
         120.327           3.378         150.409           3.383
         180.491           3.389         210.572           3.397
         240.654           3.406         270.736           3.416
         300.818           3.429         330.899           3.443
         360.981            3.46         391.063           3.479
         421.145             3.5         451.226           3.525
         481.308           3.553          511.39           3.585
         541.472           3.622         571.554           3.664
         601.635           3.713         631.717           3.769
         661.799           3.832         691.881           3.905
         721.962           3.989         739.879           4.045
         739.939           4.045
BC User HTab Sub Curve(D)= 26
              0.           3.574          31.967           3.574
          63.934           3.576          95.901           3.578
         127.868           3.582         159.835           3.587
         191.802           3.593         223.769           3.601
         255.736           3.609         287.704            3.62
         319.671           3.632         351.638           3.646
         383.605           3.662         415.572           3.681
         447.539           3.702         479.506           3.726
         511.473           3.754          543.44           3.785
         575.407           3.821         607.374           3.862
         639.341            3.91         671.308           3.964
         703.275           4.027         735.242           4.098
          767.21            4.18         798.211           4.268
BC User HTab Sub Curve(D)= 27
              0.           3.778          33.883           3.778
          67.766            3.78         101.649           3.783
         135.532           3.786         169.415           3.791
         203.298           3.797         237.181           3.804
         271.063           3.813         304.946           3.823
         338.829           3.835         372.712           3.848
         406.595           3.865         440.478           3.883
         474.361           3.904         508.244           3.927
         542.127           3.954          576.01           3.985
         609.893            4.02         643.776           4.061
         677.659           4.106         711.542           4.159
         745.425            4.22         779.307            4.29
          813.19           4.368         847.073           4.459
         849.194           4.459
BC User HTab Sub Curve(D)= 27
              0.           3.982           35.83           3.983
           71.66           3.984          107.49           3.987
          143.32            3.99          179.15           3.995
          214.98           4.001          250.81           4.008
          286.64           4.017         322.471           4.027
         358.301           4.038         394.131           4.051
         429.961           4.066         465.791           4.085
         501.621           4.105         537.451           4.128
         573.281           4.154         609.111           4.184
         644.941           4.219         680.771           4.258
         716.601           4.303         752.431           4.354
         788.261           4.413         824.091           4.481
         859.921           4.556         895.751           4.644
         916.611           4.703
BC User HTab Sub Curve(D)= 28
              0.           4.187          37.806           4.187
          75.611           4.188         113.417           4.191
         151.223           4.195         189.028           4.199
         226.834           4.205          264.64           4.212
         302.445            4.22         340.251            4.23
         378.057           4.241         415.862           4.254
         453.668           4.269         491.474           4.286
         529.279           4.306         567.085           4.329
         604.891           4.354         642.696           4.383
         680.502           4.417         718.308           4.455
         756.113           4.498         793.919           4.548
         831.725           4.605          869.53            4.67
         907.336           4.744         945.142           4.828
         982.947           4.927         982.976           4.927
BC User HTab Sub Curve(D)= 28
              0.           4.391          39.829           4.391
          79.659           4.393         119.488           4.395
         159.317           4.399         199.146           4.403
         238.976           4.409         278.805           4.416
         318.634           4.424         358.463           4.433
         398.293           4.444         438.122           4.457
         477.951           4.471         517.781           4.488
          557.61           4.508         597.439           4.529
         637.268           4.554         677.098           4.582
         716.927           4.615         756.756           4.651
         796.585           4.693         836.415           4.741
         876.244           4.797         916.073           4.858
         955.903            4.93         995.732           5.012
        1035.561           5.108        1037.798           5.108
BC User HTab Sub Curve(D)= 28
              0.           4.595          41.896           4.596
          83.792           4.597         125.688           4.599
         167.584           4.603          209.48           4.607
         251.376           4.613         293.272           4.619
         335.168           4.627         377.064           4.637
         418.959           4.647         460.855            4.66
         502.751           4.673         544.647            4.69
         586.543           4.708         628.439            4.73
         670.335           4.754         712.231           4.781
         754.127           4.812         796.023           4.848
         837.919           4.888         879.815           4.933
         921.711           4.986         963.607           5.047
        1005.503           5.116        1047.399           5.196
        1089.295           5.288        1120.183           5.365
BC User HTab Sub Curve(D)= 28
              0.           4.799          43.984             4.8
          87.968           4.801         131.953           4.804
         175.937           4.807         219.921           4.811
         263.905           4.817         307.889           4.823
         351.874           4.831         395.858            4.84
         439.842            4.85         483.826           4.862
          527.81           4.876         571.795           4.892
         615.779            4.91         659.763            4.93
         703.747           4.953         747.731            4.98
         791.716           5.009           835.7           5.043
         879.684           5.082         923.668           5.126
         967.653           5.178        1011.637           5.235
        1055.621           5.302        1099.605           5.379
        1143.589           5.468        1181.292           5.551
BC User HTab Sub Curve(D)= 29
              0.           5.004          46.104           5.004
          92.209           5.005         138.313           5.008
         184.418           5.011         230.522           5.015
         276.627            5.02         322.731           5.027
         368.836           5.034          414.94           5.043
         461.044           5.053         507.149           5.065
         553.253           5.078         599.358           5.094
         645.462           5.111         691.567            5.13
         737.671           5.152         783.775           5.178
          829.88           5.207         875.984           5.239
         922.089           5.276         968.193           5.319
        1014.298           5.367        1060.402           5.423
        1106.507           5.487        1152.611           5.561
        1198.715           5.646         1244.82           5.749
        1246.665           5.749
BC User HTab Sub Curve(D)= 30
              0.           5.208          48.232           5.208
          96.464            5.21         144.697           5.212
         192.929           5.215         241.161           5.219
         289.393           5.225         337.625           5.231
         385.858           5.238          434.09           5.247
         482.322           5.257         530.554           5.268
         578.786           5.281         627.018           5.296
         675.251           5.313         723.483           5.332
         771.715           5.354         819.947           5.378
          868.18           5.405         916.412           5.437
         964.644           5.472        1012.876           5.513
        1061.108           5.561         1109.34           5.616
        1157.573            5.68        1205.805           5.757
        1254.037           5.851        1302.269           5.966
        1350.501           6.093        1352.347           6.093
BC User HTab Sub Curve(D)= 30
              0.           5.412           50.43           5.413
         100.859           5.414         151.289           5.416
         201.718            5.42         252.148           5.424
         302.577           5.429         353.007           5.435
         403.437           5.443         453.866           5.451
         504.296           5.461         554.725           5.472
         605.155           5.485         655.585           5.501
         706.014           5.517         756.444           5.536
         806.873           5.558         857.303           5.582
         907.732           5.609         958.162            5.64
        1008.592           5.677        1059.021           5.718
        1109.451           5.768         1159.88           5.828
         1210.31           5.899         1260.74           5.983
        1311.169           6.081        1361.599           6.196
        1412.028           6.327        1450.694           6.437
BC User HTab Sub Curve(D)= 30
              0.           5.616          52.627           5.617
         105.254           5.618         157.881           5.621
         210.508           5.624         263.135           5.628
         315.762           5.633         368.389            5.64
         421.016           5.647         473.643           5.655
          526.27           5.665         578.897           5.677
         631.524            5.69         684.151           5.705
         736.778           5.721         789.405            5.74
         842.032           5.762         894.659           5.787
         947.286           5.816         999.913           5.849
         1052.54            5.89        1105.167           5.934
        1157.794           5.989        1210.421           6.052
        1263.048           6.126        1315.674           6.212
        1368.301           6.312        1420.928            6.43
        1473.555           6.564        1515.975           6.683
BC User HTab Sub Curve(D)= 31
              0.           5.821          54.869           5.821
         109.737           5.823         164.606           5.825
         219.475           5.828         274.344           5.832
         329.212           5.837         384.081           5.844
          438.95           5.851         493.818            5.86
         548.687            5.87         603.556           5.882
         658.425           5.895         713.293           5.911
         768.162           5.928         823.031           5.948
           877.9           5.972         932.768           5.999
         987.637           6.029        1042.506           6.064
        1097.374           6.105        1152.243           6.153
        1207.112           6.208        1261.981           6.273
        1316.849           6.349        1371.718           6.439
        1426.587           6.543        1481.455           6.665
        1536.324           6.803        1568.593           6.893
        1571.675           6.893
BC User HTab Sub Curve(D)= 30
              0.           6.025          57.138           6.026
         114.275           6.027         171.413           6.029
          228.55           6.033         285.688           6.037
         342.825           6.042         399.963           6.049
           457.1           6.057         514.238           6.066
         571.375           6.076         628.513           6.088
          685.65           6.102         742.788           6.118
         799.925           6.137         857.063           6.158
         914.201           6.182         971.338            6.21
        1028.476           6.241        1085.613           6.278
        1142.751            6.32        1199.888            6.37
        1257.026           6.427        1314.163           6.495
        1371.301           6.574        1428.438           6.666
        1485.576           6.774        1542.713           6.898
        1599.851           7.043         1651.07           7.186
BC User HTab Sub Curve(D)= 30
              0.           6.229          59.406            6.23
         118.813           6.231         178.219           6.234
         237.625           6.237         297.032           6.242
         356.438           6.247         415.845           6.254
         475.251           6.262         534.657           6.271
         594.064           6.282          653.47           6.294
         712.876           6.309         772.283           6.326
         831.689           6.345         891.095           6.367
         950.502           6.392        1009.908            6.42
        1069.315           6.453        1128.721           6.491
        1188.127           6.535        1247.534           6.586
         1306.94           6.646        1366.346           6.716
        1425.753           6.797        1485.159           6.893
        1544.565           7.006        1603.972           7.132
        1663.378           7.283        1718.158           7.434
BC User HTab Sub Curve(D)= 30
              0.           6.434          61.734           6.434
         123.468           6.436         185.202           6.438
         246.935           6.442         308.669           6.446
         370.403           6.452         432.137           6.459
         493.871           6.467         555.605           6.477
         617.339           6.488         679.072           6.501
         740.806           6.516          802.54           6.533
         864.274           6.553         926.008           6.576
         987.742           6.602        1049.476           6.631
         1111.21           6.666        1172.943           6.705
        1234.677           6.751        1296.411           6.804
        1358.145           6.866        1419.879           6.938
        1481.613           7.023        1543.347           7.123
         1605.08           7.239        1666.814           7.371
        1728.548           7.525        1787.566           7.688
BC User HTab Sub Curve(D)= 31
              0.           6.638          64.064           6.638
         128.129            6.64         192.193           6.643
         256.258           6.646         320.322           6.651
         384.386           6.657         448.451           6.664
         512.515           6.673          576.58           6.682
         640.644           6.694         704.708           6.707
         768.773           6.723         832.837           6.741
         896.901           6.762         960.966           6.785
         1025.03           6.812        1089.095           6.842
        1153.159           6.878        1217.223           6.919
        1281.288           6.966        1345.352           7.022
        1409.417           7.085        1473.481           7.161
        1537.545           7.249         1601.61           7.352
        1665.674           7.472        1729.738           7.608
        1793.803           7.768        1857.867           7.943
        1857.887           7.943
BC User HTab Sub Curve(D)= 45
              0.           6.842          44.175           6.842
           88.35           6.843         132.526           6.844
         176.701           6.846         220.876           6.848
         265.051           6.851         309.226           6.854
         353.402           6.857         397.577           6.862
         441.752           6.866         485.927           6.872
         530.102           6.878         574.277           6.884
         618.453           6.892         662.628             6.9
         706.803           6.909         750.978           6.919
         795.153           6.929         839.329           6.942
         883.504           6.955         927.679           6.969
         971.854           6.984        1016.029           7.001
        1060.205           7.021         1104.38            7.04
        1148.555           7.064         1192.73           7.089
        1236.905           7.116        1281.081           7.146
        1325.256            7.18        1369.431           7.217
        1413.606           7.257        1457.781           7.303
        1501.957           7.352        1546.132           7.406
        1590.307           7.469        1634.482           7.536
        1678.657           7.611        1722.832           7.695
        1767.008           7.786        1811.183           7.887
        1855.358           7.997        1899.533           8.117
         1933.48           8.217
BC User HTab Sub Curve(D)= 47
              0.           7.046          44.175           7.047
           88.35           7.047         132.526           7.048
         176.701            7.05         220.876           7.052
         265.051           7.055         309.226           7.058
         353.402           7.061         397.577           7.065
         441.752            7.07         485.927           7.075
         530.102            7.08         574.277           7.087
         618.453           7.094         662.628           7.102
         706.803            7.11         750.978           7.119
         795.153           7.129         839.329           7.141
         883.504           7.153         927.679           7.166
         971.854           7.181        1016.029           7.197
        1060.205           7.214         1104.38           7.233
        1148.555           7.254         1192.73           7.276
        1236.905           7.302        1281.081           7.329
        1325.256            7.36        1369.431           7.393
        1413.606           7.428        1457.781            7.47
        1501.957           7.512        1546.132           7.563
        1590.307           7.615        1634.482           7.677
        1678.657            7.74        1722.832           7.814
        1767.008           7.894        1811.183           7.982
        1855.358           8.078        1899.533           8.183
        1943.708           8.297        1987.884           8.421
          1990.7           8.421
BC User HTab Sub Curve(D)= 49
              0.           7.251          44.175           7.251
           88.35           7.252         132.526           7.253
         176.701           7.254         220.876           7.256
         265.051           7.259         309.226           7.261
         353.402           7.265         397.577           7.269
         441.752           7.273         485.927           7.278
         530.102           7.283         574.277           7.289
         618.453           7.296         662.628           7.303
         706.803           7.311         750.978            7.32
         795.153            7.33         839.329           7.341
         883.504           7.352         927.679           7.365
         971.854           7.378        1016.029           7.393
        1060.205           7.409         1104.38           7.426
        1148.555           7.446         1192.73           7.468
        1236.905           7.489        1281.081           7.516
        1325.256           7.542        1369.431           7.573
        1413.606           7.605        1457.781           7.643
        1501.957            7.68        1546.132           7.725
        1590.307           7.772        1634.482           7.825
        1678.657           7.883        1722.832           7.947
        1767.008           8.017        1811.183           8.094
        1855.358           8.179        1899.533           8.271
        1943.708           8.372        1987.884           8.481
        2032.059           8.598        2076.234           8.726
        2076.624           8.726
BC User HTab Sub Curve(D)= 50
              0.           7.455          44.175           7.455
           88.35           7.456         132.526           7.457
         176.701           7.458         220.876            7.46
         265.051           7.463         309.226           7.465
         353.402           7.468         397.577           7.472
         441.752           7.476         485.927           7.481
         530.102           7.486         574.277           7.492
         618.453           7.498         662.628           7.505
         706.803           7.513         750.978           7.521
         795.153           7.531         839.329           7.541
         883.504           7.552         927.679           7.564
         971.854           7.576        1016.029            7.59
        1060.205           7.605         1104.38           7.622
        1148.555           7.639         1192.73           7.659
        1236.905            7.68        1281.081           7.704
        1325.256           7.728        1369.431           7.757
        1413.606           7.786        1457.781           7.818
        1501.957           7.855        1546.132           7.893
        1590.307           7.935        1634.482           7.982
        1678.657           8.034        1722.832           8.091
        1767.008           8.153        1811.183           8.221
        1855.358           8.296        1899.533           8.377
        1943.708           8.466        1987.884           8.562
        2032.059           8.666        2076.234           8.778
        2120.409           8.899        2150.198           8.986
BC User HTab Sub Curve(D)= 50
              0.           7.659          44.175            7.66
           88.35            7.66         132.526           7.661
         176.701           7.663         220.876           7.664
         265.051           7.667         309.226           7.669
         353.402           7.672         397.577           7.676
         441.752            7.68         485.927           7.684
         530.102           7.689         574.277           7.695
         618.453           7.701         662.628           7.708
         706.803           7.715         750.978           7.723
         795.153           7.732         839.329           7.742
         883.504           7.752         927.679           7.763
         971.854           7.775        1016.029           7.788
        1060.205           7.802         1104.38           7.817
        1148.555           7.834         1192.73           7.852
        1236.905           7.872        1281.081           7.893
        1325.256           7.917        1369.431           7.942
        1413.606           7.969        1457.781           7.999
        1501.957           8.031        1546.132           8.066
        1590.307           8.105        1634.482           8.147
        1678.657           8.193        1722.832           8.244
        1767.008           8.299        1811.183            8.36
        1855.358           8.426        1899.533           8.498
        1943.708           8.576        1987.884           8.661
        2032.059           8.753        2076.234           8.853
        2120.409           8.959        2164.584           9.075
BC User HTab Sub Curve(D)= 49
              0.           7.864          44.175           7.864
           88.35           7.864         132.526           7.865
         176.701           7.867         220.876           7.868
         265.051           7.871         309.226           7.873
         353.402           7.876         397.577            7.88
         441.752           7.883         485.927           7.888
         530.102           7.893         574.277           7.898
         618.453           7.904         662.628            7.91
         706.803           7.917         750.978           7.925
         795.153           7.933         839.329           7.942
         883.504           7.952         927.679           7.963
         971.854           7.974        1016.029           7.986
        1060.205              8.         1104.38           8.014
        1148.555            8.03         1192.73           8.047
        1236.905           8.065        1281.081           8.085
        1325.256           8.106        1369.431           8.129
        1413.606           8.155        1457.781           8.183
        1501.957           8.212        1546.132           8.244
        1590.307           8.279        1634.482           8.317
        1678.657           8.359        1722.832           8.404
        1767.008           8.454        1811.183           8.508
        1855.358           8.567        1899.533           8.631
        1943.708             8.7        1987.884           8.776
        2032.059           8.857        2076.234           8.945
        2120.409           9.041
BC User HTab Sub Curve(D)= 49
              0.           8.068          43.274           8.068
          86.547           8.069         129.821            8.07
         173.095           8.071         216.368           8.072
         259.642           8.074         302.916           8.077
         346.189           8.079         389.463           8.083
         432.737           8.086          476.01            8.09
         519.284           8.095         562.558           8.099
         605.831           8.105         649.105           8.111
         692.379           8.117         735.652           8.124
         778.926           8.131         822.199            8.14
         865.473           8.149         908.747           8.158
          952.02           8.169         995.294            8.18
        1038.568           8.192        1081.841           8.205
        1125.115           8.218        1168.389           8.233
        1211.662           8.249        1254.936           8.267
         1298.21           8.285        1341.483           8.305
        1384.757           8.327        1428.031           8.351
        1471.304           8.376        1514.578           8.403
        1557.852           8.432        1601.125           8.465
        1644.399             8.5        1687.673           8.538
        1730.946           8.579         1774.22           8.623
        1817.494           8.671        1860.767           8.723
        1904.041            8.78        1947.315           8.841
        1990.588           8.908        2033.862           8.979
        2077.136           9.056
BC User HTab Sub Curve(D)= 48
              0.           8.272          42.391           8.272
          84.781           8.273         127.172           8.274
         169.562           8.275         211.953           8.276
         254.343           8.278         296.734            8.28
         339.124           8.283         381.515           8.286
         423.905           8.289         466.296           8.293
         508.686           8.297         551.077           8.301
         593.467           8.306         635.858           8.312
         678.248           8.318         720.639           8.324
         763.029           8.331          805.42           8.338
          847.81           8.346         890.201           8.355
         932.591           8.364         974.982           8.374
        1017.373           8.385        1059.763           8.397
        1102.154           8.409        1144.544           8.422
        1186.935           8.436        1229.325           8.452
        1271.716           8.468        1314.106           8.486
        1356.497           8.505        1398.887           8.525
        1441.278           8.547        1483.668            8.57
        1526.059           8.595        1568.449           8.622
         1610.84           8.652         1653.23           8.683
        1695.621           8.718        1738.011           8.755
        1780.402           8.795        1822.792           8.838
        1865.183           8.885        1907.573           8.935
        1949.964           8.989        1992.355           9.048
BC User HTab Sub Curve(D)= 46
              0.           8.476           40.66           8.477
          81.321           8.477         121.981           8.478
         162.641           8.479         203.301            8.48
         243.962           8.482         284.622           8.484
         325.282           8.486         365.943           8.489
         406.603           8.492         447.263           8.495
         487.924           8.498         528.584           8.502
         569.244           8.507         609.904           8.511
         650.565           8.517         691.225           8.522
         731.885           8.528         772.546           8.534
         813.206           8.541         853.866           8.549
         894.527           8.557         935.187           8.565
         975.847           8.575        1016.507           8.584
        1057.168           8.595        1097.828           8.606
        1138.488           8.618        1179.149           8.631
        1219.809           8.645        1260.469           8.659
        1301.129           8.675         1341.79           8.691
         1382.45           8.709         1423.11           8.728
        1463.771           8.749        1504.431            8.77
        1545.091           8.793        1585.751           8.819
        1626.412           8.845        1667.072           8.873
        1707.732           8.904        1748.393           8.937
        1789.053           8.973        1829.713           9.011
BC User HTab Sub Curve(D)= 44
              0.           8.681          37.341           8.681
          74.682           8.681         112.023           8.682
         149.364           8.683         186.705           8.684
         224.047           8.685         261.388           8.687
         298.729           8.689          336.07           8.691
         373.411           8.693         410.752           8.696
         448.093           8.699         485.434           8.702
         522.775           8.705         560.116           8.709
         597.457           8.713         634.798           8.718
          672.14           8.722         709.481           8.727
         746.822           8.733         784.163           8.739
         821.504           8.745         858.845           8.751
         896.186           8.758         933.527           8.766
         970.868           8.774        1008.209           8.783
         1045.55           8.792        1082.892           8.801
        1120.233           8.811        1157.574           8.822
        1194.915           8.833        1232.256           8.846
        1269.597           8.859        1306.938           8.872
        1344.279           8.887         1381.62           8.902
        1418.961           8.919        1456.302           8.936
        1493.643           8.954        1530.984           8.974
        1568.326           8.995        1605.667           9.017
BC User HTab Sub Curve(D)= 34
              0.           8.885          32.769           8.885
          65.537           8.885          98.306           8.886
         131.075           8.886         163.844           8.887
         196.612           8.888         229.381           8.889
          262.15           8.891         294.918           8.892
         327.687           8.894         360.456           8.896
         393.225           8.898         425.993           8.901
         458.762           8.903         491.531           8.906
         524.299           8.909         557.068           8.912
         589.837           8.916         622.605           8.919
         655.374           8.923         688.143           8.927
         720.912           8.932          753.68           8.936
         786.449           8.941         819.218           8.947
         851.986           8.952         884.755           8.958
         917.524           8.964         950.293           8.971
         983.061           8.977         1015.83           8.985
        1048.599           8.992        1081.367              9.
